HEC-RAS study NFCRNBRYRV.prj: NFCRNBRYRV

--- NFCRNBRYRV.g01 (geometry) --- (continued)

Type RM Length L Ch R = 1 ,13712   ,246.7,213.1,161.4
XS GIS Cut Line= 4
2171217.59481749459188.0196114382171287.87251115459242.870494296
2171373.57701562 459304.577737512171430.14198856459345.715899653
#Sta/Elev= 30
       0 3511.77     8.4 3508.15    18.5 3504.98    36.9 3494.08    48.3 3486.13
    64.2 3474.11    74.3 3467.13    89.5 3457.98   102.5 3448.85   108.2 3444.38
   111.1 3441.65   119.7 3432.95     124 3427.82  126.623425.789     129 3424.86
   147.9 3424.69   156.9 3424.99     161 3425.79   173.3  3429.1   182.1 3430.19
     198 3430.17   222.7 3430.81   229.8 3430.61   234.3 3431.04   237.5 3432.06
   242.5 3435.02   248.6 3440.19   254.3 3444.16   262.3 3448.98   264.7 3451.04
#Mann= 5 ,-1,0
       0      .1       0  119.15     .12       0  126.62    .045       0
     161     .08       0  244.76     .06       0
#XS Ineff= 2 , 0
                          214.19         3438.94
Permanent Ineff=
       F       F
Bank Sta=126.62,161
XS Rating Curve= 0 ,0
Exp/Cntr(USF)=0,0
Exp/Cntr=0.3,0.1

Type RM Length L Ch R = 1 ,13499   ,359.3,395.3,435.1
XS GIS Cut Line= 4
2171073.27883001459494.8499642822171190.23507961459541.632464122
2171313.68889863459405.1835062562171390.36021781459438.970867251
#Sta/Elev= 30
       0 3477.61    11.7 3472.46    19.4 3470.07    27.8 3464.94    46.2 3455.56
    63.4 3443.37      72 3435.97    80.7 3429.62    93.6 3424.77   110.8 3423.61
   124.7  3427.4   181.5 3428.16   194.4 3428.91   198.5 3427.13   204.1 3422.22
   207.5 3420.06   212.9 3418.87   245.2 3420.35   254.1 3420.65   257.9 3421.82
   263.6 3427.49   266.8 3429.79   311.9 3429.72     321 3429.09   330.2 3432.43
   351.3 3447.92   360.4 3452.08   369.5 3453.78   378.3 3453.12   393.8 3453.43
#Mann= 5 ,-1,0
       0     .12       0  155.97      .1       0   207.5    .045       0
   245.2      .1       0  305.97     .06       0
#XS Ineff= 2 , 0
          192.74 3430.47
Permanent Ineff=
       F       F
Bank Sta=207.5,245.2
XS Rating Curve= 0 ,0
Exp/Cntr(USF)=0,0
Exp/Cntr=0.3,0.1

Type RM Length L Ch R = 1 ,13103   ,326.3,345.1,352.5
XS GIS Cut Line= 4
2170936.07437531   459626.8780972171173.49299358459805.566846539
2171323.44159459459874.2932886692171395.91675175459889.288148771
#Sta/Elev= 30
       0 3472.72    20.2 3458.67      36 3445.28    50.3 3434.44    69.8 3422.42
    75.2  3420.8    87.4 3422.94   115.3 3421.46   184.5 3423.13   205.4  3422.1
   230.2  3423.7   304.5 3425.12   313.3  3423.7   326.5 3416.31  332.583413.805
   335.3 3412.57   339.7 3412.08   361.7 3412.38  374.883413.807   401.3 3415.58
   422.6 3414.49   432.1 3416.52   437.7 3419.08   462.8 3434.41     471 3440.52
   491.4 3453.61     499  3457.6   511.9 3465.68   524.1  3471.6   536.1 3475.66
#Mann= 6 ,-1,0
       0      .1       0      60     .06       0     220      .1       0
  332.58    .045       0  374.88     .12       0  427.15      .1       0
Bank Sta=332.58,374.88
XS Rating Curve= 0 ,0
Exp/Cntr(USF)=0,0
Exp/Cntr=0.3,0.1

Type RM Length L Ch R = 1 ,12758   ,274.4,281.5,282.1
XS GIS Cut Line= 4
2170851.10350141459769.329267961 2171057.2828278460030.489748056
2171163.49642018460189.1853507942171237.22114901460282.903226426
#Sta/Elev= 30
       0  3460.5    25.3 3447.75    49.1 3430.82    63.3 3422.31    81.3 3415.46
    91.8  3414.9     105 3416.46   137.4 3415.12     176 3418.53   242.7 3416.62
   325.3 3420.31     336 3418.82   348.3 3411.33   352.3 3409.84   364.9 3410.85
   417.8 3410.58     429 3411.62   441.9 3410.98  453.333408.446   470.7 3406.73
   485.2 3407.04  492.743408.446   496.2 3410.27   517.7 3429.32     527  3435.7
   535.6 3440.17   554.2 3446.69   564.4 3448.68   589.9 3458.58   642.9 3473.39
#Mann= 6 ,-1,0
       0     .06       0     120      .1       0  362.74     .12       0
  453.33    .045       0  492.74     .12       0   603.7      .1       0
#XS Ineff= 2 , 0
          354.65 3422.24
Permanent Ineff=
       F       F
Bank Sta=453.33,492.74
XS Rating Curve= 0 ,0
Exp/Cntr(USF)=0,0
Exp/Cntr=0.3,0.1

Type RM Length L Ch R = 1 ,12477   ,346.5,346.8,346.2
XS GIS Cut Line= 4
 2170696.1566137459894.2864354712170846.10521471460171.691347342
2170912.33251349460314.1425183032170987.30681399460450.345830889
#Sta/Elev= 30
       0  3432.4    12.4 3423.83    30.6 3414.39    42.1 3410.28    48.8 3409.48
    67.1 3409.62    81.8 3411.65   126.1 3411.74   139.7 3414.29   167.4 3410.52
   203.4 3412.38     217 3411.29   235.3 3413.34   269.2 3410.44   309.1 3411.15
   321.4 3406.96   330.2 3406.87   342.1 3403.56   356.7 3404.39  367.54 3402.41
   387.3 3400.92  407.653402.409   450.5 3407.05   483.4 3406.98   492.2 3409.45
   509.9 3418.16     517 3420.31   594.6 3423.83   612.9 3425.61   627.9 3429.65
#Mann= 5 ,-1,0
       0      .1       0      50     .06       0     180      .1       0
  367.54    .045       0  407.65      .1       0
#XS Ineff= 2 , 0
                          452.04         3409.07
Permanent Ineff=
       F       F
Bank Sta=367.54,407.65
XS Rating Curve= 0 ,0
Exp/Cntr(USF)=0,0
Exp/Cntr=0.3,0.1

Type RM Length L Ch R = 1 ,12130   ,182.8,181,177.3
XS GIS Cut Line= 4
2170488.72771563460196.6827808442170527.46443756460287.901513126
2170593.69173634 460406.610822262170697.40618537460581.550856774
#Sta/Elev= 30
       0 3427.51     4.9 3425.93    21.3 3418.39      44 3411.91    52.7 3410.22
    70.1  3411.9    74.4 3410.86    78.8 3408.26    82.3 3407.03    96.1  3405.9
   106.4 3401.94   118.2 3395.34  121.633394.255     128 3393.25   138.8 3392.69
   144.7 3393.16  148.413394.255   156.4 3397.75   165.2 3399.02   187.6 3399.87
   205.9 3399.36   247.7 3401.68   282.5 3402.24   321.7 3402.07   335.7 3403.72
     345 3406.79   358.9 3409.79   391.5 3411.47   419.4 3410.78   438.4 3411.92
#Mann= 6 ,-1,0
       0      .1       0      60     .06       0  121.63    .045       0
  148.41     .06       0   169.1      .1       0  285.04     .12       0
#XS Ineff= 2 , 0
                          188.67         3402.97
Permanent Ineff=
       F       F
Bank Sta=121.63,148.41
XS Rating Curve= 0 ,0
Exp/Cntr(USF)=0,0
Exp/Cntr=0.3,0.1

Type RM Length L Ch R = 1 ,11949   ,240.9,235.1,226
XS GIS Cut Line= 4
2170310.03896609460282.9032264262170350.02525969460344.132238506
 2170415.0029868460439.0996858132170561.20287278460669.020874031
#Sta/Elev= 30
       0  3437.3    33.2  3427.4    55.2 3413.69      61 3411.32    69.6 3410.22
    74.4 3408.51      84 3404.09    89.8 3400.22    98.2 3395.71   110.93392.105
   118.6 3390.82   127.7 3390.46   142.3  3390.7  146.863392.106   156.8 3395.61
   161.9 3396.74   223.8 3394.13   248.5 3393.59     257 3393.61   266.5 3394.81
   285.5 3395.72   309.7 3404.32   313.9 3405.42   318.6 3405.73   338.3 3404.59
   376.7 3404.83   389.8 3404.29     405 3405.41   441.9  3405.2   460.7  3406.1
#Mann= 7 ,-1,0
       0      .1       0      30     .06       0   110.9    .045       0
  146.86     .06       0   198.2      .1       0   388.2     .12       0
   438.2      .1       0
#XS Ineff= 2 , 0
                          162.82         3399.55
Permanent Ineff=
       F       F
Bank Sta=110.9,146.86
XS Rating Curve= 0 ,0
Exp/Cntr(USF)=0,0
Exp/Cntr=0.3,0.1

Type RM Length L Ch R = 1 ,11714   ,432.4,434.1,428.6
XS GIS Cut Line= 4
2170100.11092467460461.5919759652170156.34165005460495.330411192
2170272.55181584460576.5525700732170517.46786416460743.995174536
#Sta/Elev= 30
       0 3453.35    14.1 3446.32    22.5 3440.84    43.5 3426.04    52.2 3420.67
    65.6  3410.1    84.9 3395.95    94.7 3390.04    98.13389.052   101.3 3388.53
   119.1 3388.08     130 3388.82   175.9 3390.17   190.3  3391.9   226.3 3392.63
   245.7 3390.17   279.6 3389.87   316.9 3388.84   331.3 3391.54   342.6 3394.33
   345.7 3394.61     362 3395.13   381.3 3394.39   385.7 3394.79   405.6 3398.37
   414.7 3398.34   435.3 3399.25   449.4 3400.39   487.9  3401.1     504 3402.56
#Mann= 5 ,-1,0
       0     .12       0      40     .08       0    98.1    .045       0
     130     .08       0  155.58      .1       0
#XS Ineff= 2 , 0
                          281.06         3401.66
Permanent Ineff=
       F       F
Bank Sta=98.1,130
XS Rating Curve= 0 ,0
Exp/Cntr(USF)=0,0
Exp/Cntr=0.3,0.1

Type RM Length L Ch R = 1 ,11280   ,292.8,293.2,290.9
XS GIS Cut Line= 4
2169976.40332884460853.9574819452170076.36906285460910.188207324
2170197.57751533460977.6650777792170412.50384345461102.622245289
#Sta/Elev= 30
       0 3433.56    28.6 3417.43    45.6 3404.03    66.8 3391.43    90.3 3390.19
    96.1 3386.87   100.7 3385.44   119.1 3383.57   137.4 3383.09  155.073379.569
   160.3 3378.61     174 3378.35   184.4 3378.54  188.53 3379.57   196.2 3384.62
   201.5 3385.44   247.2 3383.55   261.1 3385.97   278.4 3386.41   302.7 3385.24
   316.6 3386.18   335.1 3383.31   353.6 3382.57   376.7 3383.64   395.4 3383.34
   418.4 3385.12   441.5 3383.81   473.9 3390.36   492.4 3400.53     502 3404.67
#Mann= 5 ,-1,0
       0      .1       0      70     .06       0  155.07    .045       0
  188.53     .12       0  293.42      .1       0
#XS Ineff= 2 , 0
                          201.98         3390.26
Permanent Ineff=
       F       F
Bank Sta=155.07,188.53
XS Rating Curve= 0 ,0
Exp/Cntr(USF)=0,0
Exp/Cntr=0.3,0.1

Type RM Length L Ch R = 1 ,10987   ,397,403.6,409.9
XS GIS Cut Line= 4
2169857.69401971461113.8683903652169936.41703524461162.601685693
2170033.88362589461206.3366943222170263.80481411461342.540006907
#Sta/Elev= 30
       0 3405.71    12.9 3402.03    31.1 3393.07      42 3388.72      50 3384.37
    56.5 3381.71    64.1 3380.29    73.9 3379.62    94.4 3380.36   105.5  3379.3
   114.2 3372.99   118.6 3372.15   127.4 3372.03   139.7 3372.94   153.7 3373.63
   182.1 3378.25   202.1 3378.91     247 3377.72   262.5 3379.38   290.4 3377.86
   314.1 3379.76   332.3 3378.84   357.9 3378.55   364.8 3377.93   378.7  3380.2
     388 3380.08     402 3377.24   411.3 3376.27   429.9 3379.92   466.7 3402.27
#Mann= 8 ,-1,0
       0     .12       0      50     .06       0   114.2    .045       0
   139.7     .06       0  199.42     .12       0  309.42      .1       0
  429.42     .12       0  449.42      .1       0
#XS Ineff= 2 , 0
                          202.42          3381.7
Permanent Ineff=
       F       F
Bank Sta=114.2,139.7
XS Rating Curve= 0 ,0
Exp/Cntr(USF)=0,0
Exp/Cntr=0.3,0.1

Type RM Length L Ch R = 1 ,10583   ,238.4,241.2,242.9
XS GIS Cut Line= 4
2169718.99156377461403.7690189872169882.68545321461521.228756446
2169992.64776062461591.2047702512170052.62720102461628.691920504
#Sta/Elev= 30
       0 3391.49    26.1 3387.61      42 3381.37    55.6 3373.66    60.5 3371.48
    73.5 3367.87    87.9 3367.73    96.5 3366.85   113.6 3367.96   119.6 3369.03
   139.4 3369.96   163.9  3369.5   198.4 3371.37   222.2 3370.29   231.5 3368.31
  239.053365.778   245.6 3364.41   260.1 3364.17   269.6 3365.28  283.253365.776
   288.6 3368.28   298.1 3374.84   307.5 3384.29   312.6 3388.53   321.3 3392.87
   335.5 3396.81   347.4 3398.88     359 3401.98   387.9 3408.11   402.5 3412.41
#Mann= 8 ,-1,0
       0      .1       0      20     .06       0     140      .1       0
  221.48     .06       0  239.05    .045       0  283.25      .1       0
  381.82     .12       0  401.82      .1       0
#XS Ineff= 2 , 0
          201.32 3374.09
Permanent Ineff=
       F       F
Bank Sta=239.05,283.25
XS Rating Curve= 0 ,0
Exp/Cntr(USF)=0,0
Exp/Cntr=0.3,0.1

Type RM Length L Ch R = 1 ,10342   ,241,246.1,250.8
XS GIS Cut Line= 4
2169615.27711474461581.208196851  2169752.729999461714.912366086
2169850.19658965461791.1362382672169945.16403696461862.361823747
#Sta/Elev= 30
       0 3385.22    23.2 3377.88    29.2 3375.53    48.7 3366.26    57.1 3363.37
      60 3363.04    79.4 3364.44   102.4  3363.7   125.1  3364.5   149.1  3367.2
     176 3366.81   185.4 3365.97   201.5 3366.32   210.1 3365.63   221.5 3363.69
   227.2 3364.23   231.7 3363.81   236.8  3362.4   241.8 3359.47   246.9 3358.29
   257.1 3358.08   267.2 3358.19  276.533359.469   292.6 3365.74   335.5 3363.88
   346.9 3364.65   378.9 3377.33   412.6 3395.18   418.9 3397.34   434.2 3401.21
#Mann= 6 ,-1,0
       0     .12       0      30      .1       0      70     .06       0
  211.76      .1       0   241.8    .045       0  276.53      .1       0
#XS Ineff= 2 , 0
          154.57 3369.27  294.83         3369.73
Permanent Ineff=
       F       F
Bank Sta=241.8,276.53
XS Rating Curve= 0 ,0
Exp/Cntr(USF)=0,0
Exp/Cntr=0.3,0.1

Type RM Length L Ch R = 1 ,10096   ,293.5,297.6,301.4
XS GIS Cut Line= 4
2169537.80367088461806.1310983682169615.27711474461901.098545675
2169695.24970194462001.064279683 2169767.7248591462082.286438564
#Sta/Elev= 30
       0 3374.76    10.1 3374.02    22.7 3374.16    34.9 3373.16    49.3 3366.59
    54.4 3364.94    57.9 3364.62    69.2 3365.25    73.4 3364.84    77.8 3363.72
    86.5 3359.81    92.3 3358.23   103.4 3357.59   126.1 3358.58   142.9 3357.45
   153.4 3357.29  159.733354.465   163.1 3353.08   173.9 3352.66   185.9 3353.31
  192.453354.463   199.5 3355.62   211.5 3355.43   226.4 3357.86   240.5  3357.7
   256.1 3360.29   271.1 3361.35   310.8 3374.06   331.1 3382.46   359.4 3393.02
#Mann= 4 ,-1,0
       0     .06       0  152.56      .1       0  159.73    .045       0
  192.45      .1       0
#XS Ineff= 2 , 0
          129.81 3362.58
Permanent Ineff=
       F       F
Bank Sta=159.73,192.45
XS Rating Curve= 0 ,0
Exp/Cntr(USF)=0,0
Exp/Cntr=0.3,0.1

Type RM Length L Ch R = 1 ,9798    ,176.4,182.3,188.2
XS GIS Cut Line= 4
2169329.12520114461964.8267011052169386.60549819462073.539436839
2169447.83451027462186.0008875972169509.06352235462303.460625056
#Sta/Elev= 30
       0 3367.84    63.7 3366.71    72.8 3365.95    88.4 3360.58    91.3  3360.2
   100.2 3360.15     112 3358.24   126.3 3352.87   132.7 3349.82   140.8 3349.44
  148.053347.987   154.4 3346.96   177.2    3347   181.8 3347.34  184.063347.988
   195.4 3351.03   200.5 3351.25   218.2 3350.72   228.1 3353.11   236.4 3354.53
   250.1 3354.84   259.1 3353.36   271.4 3354.63   277.2 3356.68   290.7 3364.14
   301.1 3367.28   312.9 3369.07   346.9 3372.22   372.2 3376.08   383.5 3376.92
#Mann= 4 ,-1,0
       0     .12       0      70     .06       0  148.05    .045       0
  184.06      .1       0
Bank Sta=148.05,184.06
XS Rating Curve= 0 ,0
Exp/Cntr(USF)=0,0
Exp/Cntr=0.3,0.1

Type RM Length L Ch R = 1 ,9616    ,252,255.1,256.7
XS GIS Cut Line= 4
2169189.17317353462031.0539998852169230.40903881462141.016307294
2169267.89618906462268.4726181542169440.33708022462498.393806371
#Sta/Elev= 30
       0 3364.67    27.9 3362.68    32.2  3361.5      45 3354.77    57.8 3349.65
    96.3 3349.88   113.3 3351.14   125.9 3350.16   134.3 3347.84   146.8  3346.8
  154.243344.866   160.9 3343.84   192.7 3343.64  199.683344.866   209.3 3350.91
   213.5 3351.91     226 3349.86   238.5 3351.42   277.4 3353.47   296.2 3359.12
   321.2 3362.56   336.2 3362.97   346.2 3362.37   361.2 3367.18   373.9 3369.35
   417.4 3372.02   444.1 3372.61   476.7 3376.75   522.4  3380.4   537.7 3380.67
#Mann= 5 ,-1,0
       0      .1       0     100     .06       0  154.24    .045       0
  199.68     .06       0  207.44      .1       0
Bank Sta=154.24,199.68
XS Rating Curve= 0 ,0
Exp/Cntr(USF)=0,0
Exp/Cntr=0.3,0.1

Type RM Length L Ch R = 1 ,9361    ,247.7,244.2,238.8
XS GIS Cut Line= 4
2168976.74598876462128.5205905432168985.49299049 462159.75988242
2169016.73228237462315.9563418072169091.70658287462618.352687181
#Sta/Elev= 30
       0 3370.51    13.1 3362.46    25.6 3352.82      42 3344.58    46.1 3343.66
    82.8 3344.15   92.823341.184   100.5 3339.61   123.6 3339.99  134.053341.183
   141.3 3342.26   164.4 3341.68   168.5 3342.37   172.6 3344.03   180.7 3350.29
   188.9 3351.97   217.7 3351.71   234.2 3349.67   250.7 3349.96     263 3351.64
   279.5 3349.26   345.5 3353.83   374.3 3354.24   394.9 3352.03   407.3 3354.27
   423.8 3355.52   436.7 3354.67   459.8 3355.45   477.3 3361.89   503.3 3377.93
#Mann= 4 ,-1,0
       0     .06       0   92.44      .1       0   92.82    .045       0
  134.05      .1       0
Bank Sta=92.82,134.05
XS Rating Curve= 0 ,0
Exp/Cntr(USF)=0,0
Exp/Cntr=0.3,0.1

Type RM Length L Ch R = 1 ,9117    ,346.6,347.5,339.3
XS GIS Cut Line= 4
2168740.57694217 462223.488037852168751.82308725462265.973474803
2168795.55809587462379.684497237 2168849.2896779462652.091122408
#Sta/Elev= 30
       0  3368.1    10.9 3362.85    20.7 3354.46    30.7 3344.77    34.9 3342.28
      39 3341.01      56 3340.38    68.8 3338.28      86 3338.21   99.993336.396
   108.6  3335.1     116 3334.91   133.1 3335.11  138.313336.394   150.2 3342.28
   163.1 3343.25   183.6 3343.61   208.1  3342.5   265.2 3341.59   277.4 3341.86
   286.8 3342.87   301.8 3342.96   317.4 3341.88   342.6 3341.88   375.2 3343.37
   387.5 3345.13   395.6 3347.95   420.1  3353.4   428.2 3356.97   443.4  3366.2
#Mann= 3 ,-1,0
       0     .06       0   99.99    .045       0  138.31      .1       0
Bank Sta=99.99,138.31
XS Rating Curve= 0 ,0
Exp/Cntr(USF)=0,0
Exp/Cntr=0.3,0.1

Type RM Length L Ch R = 1 ,8769    ,237,250.9,271.2
XS GIS Cut Line= 4
2168425.68488005462224.7376095252168424.43530837462349.694777035
2168491.91217883462472.152801194 2168498.1600372462678.332127585
#Sta/Elev= 30
       0 3357.73    28.4  3348.9    32.4 3346.56    40.4 3339.78    48.4 3335.92
    56.4 3335.15    76.4    3337    96.4 3336.51   116.4 3337.42   130.3 3335.67
   139.63332.208   142.6 3330.66   149.3 3329.79   165.9 3330.36  179.113332.207
   203.9  3333.6   224.5 3332.55   230.4 3333.24   238.6 3335.69     251 3336.81
   317.8 3334.82   341.8 3337.62   353.8 3335.66   361.9 3336.02   369.9 3335.11
   381.9 3335.97   425.9  3335.4   429.9 3336.89   441.9 3344.29   471.1 3370.14
#Mann= 4 ,-1,0
       0     .06       0     100      .1       0   139.6    .045       0
  179.11      .1       0
#XS Ineff= 2 , 0
          115.51 3340.64  250.83            3342
Permanent Ineff=
       F       F
Bank Sta=139.6,179.11
XS Rating Curve= 0 ,0
Exp/Cntr(USF)=0,0
Exp/Cntr=0.3,0.1

Type RM Length L Ch R = 1 ,8518    ,222.4,221.3,220.8
XS GIS Cut Line= 4
2168346.96186451462232.2350395762168264.49013396462448.410939367
2168234.50041376462555.8741034262168249.49527386462643.344120682
#Sta/Elev= 30
       0 3355.12       6 3352.61    18.1 3344.94      31 3338.21    43.8 3334.25
    52.7 3333.15    60.9 3332.85    75.2 3335.79    89.7 3335.19      99 3335.69
   148.5 3330.58   163.7 3330.43   179.5 3331.74   189.4 3330.57     242 3329.87
   257.1 3327.67   269.5 3327.94     282 3326.83   303.7 3327.12     307 3327.39
  308.273328.223   311.1 3330.09   319.4 3332.09   339.4 3333.03   352.3 3335.58
   364.6 3336.86   372.7 3339.27   376.8 3341.22     393 3353.67   431.7 3385.84
#Mann= 3 ,-1,0
       0      .1       0   269.5    .045       0  308.27      .1       0
#XS Ineff= 2 , 0
          177.67 3337.08  326.18         3338.03
Permanent Ineff=
       F       F
Bank Sta=269.5,308.27
XS Rating Curve= 0 ,0
Exp/Cntr(USF)=0,0
Exp/Cntr=0.3,0.1

Type RM Length L Ch R = 1 ,8297    ,219.9,198.6,178
XS GIS Cut Line= 4
2168114.54153295462207.2436060742168054.56209254462383.433212262
2168010.82708391  462547.12710172168030.82023072462635.846690632
#Sta/Elev= 30
       0 3355.47    19.2 3348.86    23.2 3346.79    35.8 3337.47    44.4 3331.98
    61.2  3326.3    65.4 3325.61    73.9  3326.7      95 3326.21   116.1 3323.05
     120 3323.19   137.3 3326.18   145.2 3326.73   162.6 3324.78   183.7  3325.4
   199.3 3323.22   208.6 3321.68   233.5 3321.78   247.4 3323.72   254.2 3326.93
   264.3 3327.61   287.3  3327.9   295.6 3326.86   312.1 3327.09   332.8 3325.02
   361.8 3327.66     370  3329.1   402.8 3341.06   406.9  3343.4   446.5 3372.76
#Mann= 5 ,-1,0
       0      .1       0      20     .06       0     120      .1       0
   199.3    .045       0   247.4      .1       0
#XS Ineff= 2 , 0
          145.76 3330.45  284.42         3329.18
Permanent Ineff=
       F       F
Bank Sta=199.3,247.4
XS Rating Curve= 0 ,0
Exp/Cntr(USF)=0,0
Exp/Cntr=0.3,0.1

Type RM Length L Ch R = 1 ,8098    ,162.8,184,191.9
XS GIS Cut Line= 4
2167857.12976788462229.735896226 2167835.8870494462364.689637136
2167882.12120138462430.9169359162167934.60321173462644.593692357
#Sta/Elev= 30
       0 3341.38     3.5 3340.14    19.7 3338.13      44  3337.5    68.3 3334.86
   101.8 3334.29     129 3331.33   137.2 3329.84     140  3328.4   142.9 3326.37
   148.7 3320.91  151.383319.005   156.7 3317.94   176.2 3317.45   188.9 3318.61
   200.4 3319.13     221 3321.97   269.1 3319.31   277.4 3319.86   310.3 3319.12
   343.3 3319.16   355.6 3320.01   359.8 3321.37   363.9 3324.94   376.2 3338.52
   380.4 3341.52   392.7 3351.96   400.9 3357.89   417.4 3371.43   437.4 3385.83
#Mann= 4 ,-1,0
       0     .06       0      90      .1       0  151.38    .045       0
   188.9      .1       0
#XS Ineff= 2 , 0
                          321.88         3326.87
Permanent Ineff=
       F       F
Bank Sta=151.38,188.9
XS Rating Curve= 0 ,0
Exp/Cntr(USF)=0,0
Exp/Cntr=0.3,0.1

Type RM Length L Ch R = 1 ,7914    ,192.1,205.7,214.3
XS GIS Cut Line= 4
2167793.40161245462234.7341829262167757.16403387462445.911796017
2167778.40675235462587.1133953032167789.65289742462667.085982509
#Sta/Elev= 30
       0 3341.74    10.6 3340.59    18.7 3338.61    34.9 3337.52    63.4  3332.7
    89.7 3331.54   116.1 3328.69   132.4 3328.04   156.7 3322.84   181.1 3320.85
   193.2 3322.03   201.3 3319.88   205.4 3319.52   229.7 3319.09   240.9 3317.14
   262.1 3316.94   274.2 3314.87   286.3 3314.99  294.143313.765   310.6 3311.48
   334.9 3312.74  341.113313.767     343 3314.23   346.4 3318.14   355.1 3331.39
   363.2 3339.58   375.3 3348.07   399.7 3369.05   420.7 3382.05   437.8 3394.29
#Mann= 4 ,-1,0
       0     .06       0      90      .1       0  294.14    .045       0
  341.11      .1       0
Bank Sta=294.14,341.11
XS Rating Curve= 0 ,0
Exp/Cntr(USF)=0,0
Exp/Cntr=0.3,0.1

Type RM Length L Ch R = 1 ,7709    ,277,276.2,275.9
XS GIS Cut Line= 4
2167640.95386808462244.7307563272167588.47185773462458.407512768
 2167559.7317092462567.120248501 2167549.7351358462654.590265758
#Sta/Elev= 30
       0 3331.96     4.6  3330.6    21.1 3327.35    41.7 3326.33    62.2 3324.18
    70.5 3324.06    91.1 3319.29   111.7 3316.42   128.1 3316.61   139.9 3315.54
   152.9 3315.82   173.5 3314.47   185.8 3314.34   210.5 3314.21   231.2 3315.63
   239.4 3314.08   247.7  3310.1  251.053309.013   260.1 3307.61   268.4 3307.19
   276.7 3307.59  282.933309.013   294.5 3312.31   313.9 3324.05   350.7 3340.62
   362.8 3346.93   390.9 3359.02     399 3363.46     411 3368.95   420.5 3372.61
#Mann= 4 ,-1,0
       0     .06       0      80      .1       0  251.05    .045       0
  282.93      .1       0
#XS Ineff= 2 , 0
          228.82 3318.55
Permanent Ineff=
       F       F
Bank Sta=251.05,282.93
XS Rating Curve= 0 ,0
Exp/Cntr(USF)=0,0
Exp/Cntr=0.3,0.1

Type RM Length L Ch R = 1 ,7432    ,272.8,282.5,291.7
XS GIS Cut Line= 5
2167381.04295966462209.7427494242167319.81394759462389.681070638
2167289.82422738462524.6348115482167276.07893896462619.602258856
2167321.06351926462673.333840885
#Sta/Elev= 30
       0 3328.99     3.6 3327.72    12.8 3321.62    24.8 3314.79    33.2  3311.3
    41.7 3309.06    62.8 3307.12   113.5 3309.19   126.3 3308.51   142.1 3309.47
   172.6  3308.9   201.8 3309.57   218.2 3308.65     2303305.061   234.6 3303.64
   239.6 3303.36   275.6 3303.73   279.7 3304.21  281.263305.061   286.6 3309.13
   296.1 3319.21     300 3321.24   303.3 3322.06   316.3 3321.55   328.9 3322.53
     341 3321.37   402.6 3325.34   468.1 3328.53   474.3 3329.79   494.3 3341.18
#Mann= 5 ,-1,0
       0      .1       0      40     .06       0  220.07      .1       0
     230    .045       0  281.26      .1       0
#XS Ineff= 2 , 0
          200.77 3312.27
Permanent Ineff=
       F       F
Bank Sta=230,281.26
XS Rating Curve= 0 ,0
Exp/Cntr(USF)=0,0
Exp/Cntr=0.3,0.1

Type RM Length L Ch R = 1 ,7150    ,223.1,225.6,218.1
XS GIS Cut Line= 4
2167171.11491825462146.0145939942167146.12348475462205.994034399
2167013.66888719462405.9255024142166919.95101155462527.133954898
#Sta/Elev= 30
       0 3328.81    20.8 3316.41    33.8 3311.31    42.4 3306.87    68.7 3305.44
    83.2 3301.53   133.7 3304.68   148.2 3302.17   155.4 3301.65   189.9 3302.09
   223.23300.181   231.9 3298.97   250.5 3298.84   256.3  3298.9  260.853300.181
   279.4 3306.89   285.1 3308.17   294.3 3307.52   307.2 3309.09   322.4 3308.78
   339.3 3310.35   349.4 3309.46   366.1 3309.42   384.8 3310.88   413.7 3310.59
   420.2 3309.88   433.7  3311.1   442.2 3314.12   451.1    3321     458 3325.36
#Mann= 4 ,-1,0
       0     .06       0  194.98      .1       0   223.2    .045       0
  260.85      .1       0
#XS Ineff= 2 , 0
          135.31 3306.35
Permanent Ineff=
       F       F
Bank Sta=223.2,260.85
XS Rating Curve= 0 ,0
Exp/Cntr(USF)=0,0
Exp/Cntr=0.3,0.1

Type RM Length L Ch R = 1 ,6924    ,191.7,184.6,173.2
XS GIS Cut Line= 4
2166969.93387856462071.0402934882166944.94244506462136.018020593
2166818.73570587462387.1819272882166798.74255907462420.920362515
#Sta/Elev= 30
       0    3338     6.6 3336.71    23.7 3330.41      28 3327.51    36.6 3319.11
    45.1 3312.58      58 3305.19    62.3 3304.31    75.4 3303.38    79.9 3301.82
   87.933296.132    93.3 3294.11    97.8 3294.07   115.7 3294.59  124.713296.132
   139.6 3298.29   151.5 3301.06   178.4 3301.22   231.9 3299.41     250 3299.59
   276.8 3300.93   294.5 3299.66   308.2 3301.17   318.3 3300.57   326.1  3300.8
   330.3 3301.62   365.7 3312.38   374.5 3315.78   385.6 3321.07   389.9 3322.38
#Mann= 4 ,-1,0
       0     .06       0      60      .1       0   87.93    .045       0
  124.71      .1       0
#XS Ineff= 2 , 0
                          177.34         3304.32
Permanent Ineff=
       F       F
Bank Sta=87.93,124.71
XS Rating Curve= 0 ,0
Exp/Cntr(USF)=0,0
Exp/Cntr=0.3,0.1

Type RM Length L Ch R = 1 ,6740    ,247.6,242.4,237.7
XS GIS Cut Line= 4
2166776.25026892462019.8078548092166753.75797877 462096.03172699
2166746.26054872462189.7496026222166753.75797877462408.424645764
#Sta/Elev= 30
       0    3327    26.5  3319.6    34.8 3316.71    49.5 3309.62    59.8 3303.46
      64 3301.84    88.6 3299.55    96.4 3295.38  102.28 3293.82   104.7 3292.97
   108.7 3292.47   120.8 3292.14   144.8 3292.81  149.03 3293.82   156.9 3297.43
   160.9  3298.5   168.9 3298.89   194.1 3297.69     229 3297.72     241 3296.44
     289 3297.56     293 3298.32     301 3301.29     309 3303.05     317 3306.15
     333 3310.95     345 3315.49     357 3318.97     377 3323.52   392.3 3328.05
#Mann= 4 ,-1,0
       0      .1       0      10     .06       0  102.28    .045       0
  149.03      .1       0
#XS Ineff= 2 , 0
                           168.1         3301.39
Permanent Ineff=
       F       F
Bank Sta=102.28,149.03
XS Rating Curve= 0 ,0
Exp/Cntr(USF)=0,0
Exp/Cntr=0.3,0.1

Type RM Length L Ch R = 1 ,6497    ,213.7,230.1,248.1
XS GIS Cut Line= 4
2166580.06751593461924.8404075022166500.09492872462067.291578463
 2166521.3376472462283.4674782552166498.84535705462335.949488609
#Sta/Elev= 30
       0 3298.35       6 3296.05    16.1 3295.39    48.8 3295.75    65.1  3296.9
    92.1 3296.32   114.7 3297.21   123.6 3296.48     138 3292.76   151.8 3291.83
   177.3 3294.17   213.5 3294.58   238.4  3289.3   241.6 3288.05   245.6 3287.87
   277.8    3289   289.9 3287.74   293.9 3287.83   305.9 3292.48     310 3293.32
     318 3292.83   330.1 3290.51   358.2 3292.44   370.4 3295.29   382.8 3301.58
   395.5 3311.53   404.5 3317.63   417.3 3328.14   425.4 3336.39   437.7 3346.56
#Mann= 4 ,-1,0
       0     .06       0     120      .1       0   238.4    .045       0
   277.8      .1       0
#XS Ineff= 2 , 0
          213.42 3296.76  313.53         3296.55
Permanent Ineff=
       F       F
Bank Sta=238.4,277.8
XS Rating Curve= 0 ,0
Exp/Cntr(USF)=0,0
Exp/Cntr=0.3,0.1

Type RM Length L Ch R = 1 ,6267    ,266.3,267.4,264.4
XS GIS Cut Line= 4
 2166526.3359339 461902.348117352166356.39418609462084.785581914
2166261.42673878462164.7581691212166248.93102203462182.252172572
#Sta/Elev= 30
       0  3297.1     3.9 3295.39       9 3294.13    17.7  3293.5    25.7 3293.51
    47.6 3295.65    71.5 3294.54    80.4 3293.43    85.9 3294.15    97.1 3294.28
   120.5  3290.6   130.9 3289.51   149.9 3290.02   156.4 3290.67   185.1 3289.55
     196 3290.16   235.6 3290.05   255.4 3290.88   289.5 3285.57   322.8 3283.53
   328.1 3282.77   334.9 3282.61   343.1 3283.08   346.3 3283.71   354.8 3287.03
   364.7 3297.18   378.9 3307.57   383.8 3311.92   388.7 3315.46     395 3321.14
#Mann= 5 ,-1,0
       0      .1       0      30     .06       0     170      .1       0
   322.8    .045       0   346.3      .1       0
#XS Ineff= 2 , 0
          253.91 3293.18
Permanent Ineff=
       F       F
Bank Sta=322.8,346.3
XS Rating Curve= 0 ,0
Exp/Cntr(USF)=0,0
Exp/Cntr=0.3,0.1

Type RM Length L Ch R = 1 ,6000    ,218.7,220.6,218.2
XS GIS Cut Line= 4
2166357.64375776461794.8849532922166256.42845208461856.113965372
2166136.46957127461943.5839826282166110.22856609462033.553143235
#Sta/Elev= 30
       0 3306.74    15.7 3303.87    31.9    3299    53.1 3293.93    66.8 3291.45
    81.2 3290.33    87.2 3287.97    89.4 3287.52   109.2  3287.9   119.2 3287.11
   130.7 3285.14   138.4  3285.4   150.7 3284.88   153.6 3284.23   162.2 3278.17
     165 3277.31   176.5 3276.92   197.8 3277.88   202.8 3277.83   212.7  3279.4
   237.4  3280.9   242.4 3282.83   252.3 3290.79   255.9  3292.1   271.5 3293.16
   285.1 3295.63   301.8 3297.01   309.8 3298.58   342.5 3303.52   360.5 3309.13
#Mann= 4 ,-1,0
       0     .06       0   162.2    .045       0   197.8     .06       0
  208.29      .1       0
Bank Sta=162.2,197.8
XS Rating Curve= 0 ,0
Exp/Cntr(USF)=0,0
Exp/Cntr=0.3,0.1

Type RM Length L Ch R = 1 ,5779    ,339.5,322.7,292.6
XS GIS Cut Line= 4
 2166230.1874469461638.6884939052166151.46443137461677.425215833
2166020.25940549 461764.895233092166014.01154711461978.571989531
#Sta/Elev= 30
       0 3289.23     6.4 3286.59    12.3 3285.19    33.4 3284.35    42.4 3282.49
    72.1 3280.49    96.5 3280.74   106.1 3282.84   108.9 3282.59   110.9 3282.13
   115.7 3278.15   120.5 3275.57  150.053274.228   168.6 3272.34   173.6 3272.51
  180.083274.228   187.8  3277.4   205.3 3279.06   228.4 3279.36   257.7 3276.96
   269.7 3278.57   277.7 3278.74   285.7 3280.16   301.7 3280.92   329.7 3284.39
   341.8 3284.25   356.9 3286.31   385.8 3288.25   441.8 3295.93   459.2 3300.35
#Mann= 4 ,-1,0
       0      .1       0      50     .06       0  150.05    .045       0
  180.08      .1       0
#XS Ineff= 2 , 0
                          225.52         3281.19
Permanent Ineff=
       F       F
Bank Sta=150.05,180.08
XS Rating Curve= 0 ,0
Exp/Cntr(USF)=0,0
Exp/Cntr=0.3,0.1

Type RM Length L Ch R = 1 ,5456    ,296.7,292.6,290.4
XS GIS Cut Line= 4
2165880.30737787461421.2630224382165876.55866285 461509.98261137
 2165874.0595195461704.9157926852165907.79795473461973.573702831
#Sta/Elev= 30
       0 3292.52    19.9 3282.61    27.9 3279.97      64 3279.51      76 3275.73
      84 3276.69     100 3276.93     108 3274.75  115.423268.252     120 3266.91
   132.2 3266.65     148 3266.68   159.23268.256     172 3271.74     216 3271.11
     228 3271.75     260 3275.68     280 3275.23   296.6 3273.25   324.3 3273.04
   356.6 3270.46   380.8 3270.65   384.8 3271.42   396.9 3276.38     405 3278.08
   433.2 3277.24   461.4 3281.25   481.6 3286.76   512.1  3296.5   554.5 3308.23
#Mann= 4 ,-1,0
       0     .06       0      10      .1       0  115.42    .045       0
   159.2      .1       0
#XS Ineff= 2 , 0
                          258.75         3276.74
Permanent Ineff=
       F       F
Bank Sta=115.42,159.2
XS Rating Curve= 0 ,0
Exp/Cntr(USF)=0,0
Exp/Cntr=0.3,0.1

Type RM Length L Ch R = 1 ,5164    ,162,166,169.1
XS GIS Cut Line= 4
2165596.65460763 461375.028870462165591.65632093 461576.20991015
 2165607.9007527461724.9089394872165629.14347118461986.069419582
#Sta/Elev= 30
       0 3287.22    30.2 3287.07    46.8 3281.71    66.2 3277.25    90.2 3275.52
   126.2 3268.14   162.2 3267.04   182.2 3270.78   190.2 3270.49   198.2  3268.4
     228 3269.17   238.4 3267.56  253.753261.166   260.6 3259.95   290.7 3259.58
  300.163261.166   322.9 3269.33   347.1 3271.02   379.2 3269.31   410.7 3270.38
   451.4 3269.56   471.5 3266.69   483.5 3266.23   499.6 3263.51   531.7 3263.56
   539.7 3266.19   559.2 3278.99   585.1 3302.54   600.9 3315.91   612.8 3324.69
#Mann= 4 ,-1,0
       0     .06       0      60      .1       0  253.75    .045       0
  300.16      .1       0
#XS Ineff= 2 , 0
                          351.93         3272.79
Permanent Ineff=
       F       F
Bank Sta=253.75,300.16
XS Rating Curve= 0 ,0
Exp/Cntr(USF)=0,0
Exp/Cntr=0.3,0.1

Type RM Length L Ch R = 1 ,4998    ,199.6,221.4,237.9
XS GIS Cut Line= 4
2165514.18287707461343.7895785822165437.95900489461551.218476648
2165434.21028986461742.4029429382165310.50269403461866.110538773
#Sta/Elev= 30
       0 3277.76     2.6 3276.81      10 3278.15    18.5 3277.19      40 3265.38
    52.5 3261.73    65.4 3260.12   108.6  3260.1   133.5 3261.25   191.4 3261.76
     206  3262.9     231 3262.31     247 3263.95     283 3264.14     291  3263.4
     312  3258.3     319 3256.78   346.3 3256.71     359 3258.07     383 3264.17
     403 3264.75   452.4 3264.28   478.4 3260.92   489.2 3258.49     518 3258.58
   523.1 3259.98   528.8  3263.5   542.9 3274.67     574 3297.56   587.2 3303.87
#Mann= 4 ,-1,0
       0     .06       0     100      .1       0     312    .045       0
     359      .1       0
#XS Ineff= 2 , 0
          281.85    3267   393.4         3267.27
Permanent Ineff=
       F       F
Bank Sta=312,359
XS Rating Curve= 0 ,0
Exp/Cntr(USF)=0,0
Exp/Cntr=0.3,0.1

Type RM Length L Ch R = 1 ,4776    ,164,167,173
XS GIS Cut Line= 4
2165505.43587535461345.0391502572165357.98641768 461576.20991015
2165199.29081495461658.6816407072165171.80023809461677.425215833
#Sta/Elev= 30
       0 3276.49     4.9 3277.53    14.4 3276.36    24.2 3269.73    28.6 3267.44
    39.5 3263.44    52.4 3261.33    70.5 3260.29   158.5 3260.58   180.6 3261.31
   221.2 3259.93   241.4 3261.86   251.6 3261.14   265.9 3261.62   280.7 3260.57
   293.6  3255.5   307.8 3254.54   334.8 3258.36   348.4 3257.33   357.4 3257.48
   379.9 3255.03   411.5 3254.75   424.6 3253.74   433.5 3253.87   435.7 3254.95
     443 3258.45   448.3 3259.58   465.7 3261.22   478.8 3261.06   486.3 3261.78
#Mann= 4 ,-1,0
       0     .06       0     110      .1       0   411.5    .045       0
   435.7      .1       0
#XS Ineff= 2 , 0
          265.75 3262.94
Permanent Ineff=
       F       F
Bank Sta=411.5,435.7
XS Rating Curve= 0 ,0
Exp/Cntr(USF)=0,0
Exp/Cntr=0.3,0.1

Type RM Length L Ch R = 1 ,4609    ,201.8,188.8,158.3
XS GIS Cut Line= 4
2165494.18973027461342.5400069072165347.98984428461482.492034518
2165160.55409302461519.9791847712165120.56779942461613.697060403
#Sta/Elev= 30
       0 3275.54    11.8 3275.45    15.4 3274.27    23.1 3269.29    32.7 3264.52
    41.6 3262.22    85.8 3261.25   113.5 3257.89   144.7 3260.44   171.6    3259
   183.1 3259.75   200.5  3258.8   211.3 3259.77     243  3257.3   255.2 3251.33
   259.3 3250.51   275.2 3249.22   287.9 3250.49   300.1 3250.95   326.2 3255.02
   332.7 3254.72   340.9 3251.63   349.1 3254.25   361.3 3255.33   381.7 3253.18
   393.5 3255.11   416.1 3255.22   440.5 3258.99   452.7 3261.97   495.4 3263.91
#Mann= 4 ,-1,0
       0     .06       0     130      .1       0   259.3    .045       0
   287.9      .1       0
#XS Ineff= 2 , 0
                          362.49         3258.68
Permanent Ineff=
       F       F
Bank Sta=259.3,287.9
XS Rating Curve= 0 ,0
Exp/Cntr(USF)=0,0
Exp/Cntr=0.3,0.1

Type RM Length L Ch R = 1 ,4421    ,207.3,202.4,185.4
XS GIS Cut Line= 4
 2165261.7693987 461250.071702952165240.52668023461292.557139903
2165179.29766815461401.2698756372165110.57122601461602.450915327
#Sta/Elev= 30
       0 3291.88    12.4 3283.25    24.4 3280.44    43.7 3270.87    48.2 3266.29
    57.4 3253.07      62 3248.99    65.1 3247.75    74.6 3246.52    80.3 3246.41
    98.1 3246.52  109.863247.751   121.6 3251.23   126.3 3253.16   130.8 3254.03
   171.6 3254.27   184.9 3253.37   201.8 3254.31   214.4  3255.9   227.1 3255.87
     244 3257.21   269.4 3256.98   303.2 3254.37   319.6 3257.39   328.6 3258.28
     337 3260.78   345.5 3260.83   354.2 3261.88   373.1 3262.21   384.9 3263.26
#Mann= 3 ,-1,0
       0     .06       0    65.1    .045       0  109.86      .1       0
Bank Sta=65.1,109.86
XS Rating Curve= 0 ,0
Exp/Cntr(USF)=0,0
Exp/Cntr=0.3,0.1

Type RM Length L Ch R = 1 ,4218    ,267,258.5,244.5
XS GIS Cut Line= 4
2165046.84307059461142.6085388922165035.59692551461230.078556149
2165020.60206541461357.5348670082165068.08578906461597.452628627
#Sta/Elev= 30
       0 3295.86     6.6 3289.47    22.8 3276.99    26.8 3275.31    30.8 3275.58
    42.9 3274.34      47 3273.12      51 3270.12    75.2  3254.8    83.3 3251.32
    91.3 3248.99   115.5 3243.83   142.6 3242.91   151.7 3241.88   163.8 3241.56
   171.9 3241.66   175.9  3242.8   179.9 3246.49   183.9 3247.87     196 3248.29
   208.1 3250.38   221.7 3251.53   240.6 3251.37   253.3 3252.79   269.2 3252.83
   297.7  3254.6   371.1 3255.16   399.6 3258.22   424.1 3260.02   461.1  3261.7
#Mann= 5 ,-1,0
       0     .06       0   98.19     .12       0   142.6    .045       0
   175.9     .12       0  198.19      .1       0
Bank Sta=142.6,175.9
XS Rating Curve= 0 ,0
Exp/Cntr(USF)=0,0
Exp/Cntr=0.3,0.1

Type RM Length L Ch R = 1 ,3960    ,178.2,181.7,183
XS GIS Cut Line= 4
2164716.95614836461190.0922625452164765.68944369461288.808424878
2164813.17316734461393.7724455862164916.88761638461627.442348829
#Sta/Elev= 30
       0 3267.72    16.7  3264.2    25.6 3263.22    34.7 3259.94    43.5 3259.32
      57 3256.36    65.9 3255.62    79.3 3252.56    97.1  3253.4   101.6 3252.81
   106.7 3251.02   112.2 3247.34   123.7 3241.58  134.343237.842   141.2 3236.44
     150 3236.31   157.6 3236.51  164.123237.841   176.4 3240.92   185.1 3243.95
   189.5 3244.44   207.1 3244.24   233.4 3247.45   255.3 3245.35   303.4 3249.47
   325.3 3250.21   404.1  3251.1   429.9 3253.77     461 3259.15   480.9 3261.23
#Mann= 4 ,-1,0
       0      .1       0      50     .06       0  134.34    .045       0
  164.12      .1       0
#XS Ineff= 2 , 0
                          190.32         3246.14
Permanent Ineff=
       F       F
Bank Sta=134.34,164.12
XS Rating Curve= 0 ,0
Exp/Cntr(USF)=0,0
Exp/Cntr=0.3,0.1

Type RM Length L Ch R = 1 ,3778    ,322.6,339.3,355.7
XS GIS Cut Line= 4
2164630.73570278461212.584552697 2164594.4981242461335.042576857
2164653.22799293461481.2424628432164740.69801019461694.919219284
#Sta/Elev= 30
       0 3253.29       9 3250.41    21.5 3249.12    29.8 3247.53    46.5  3242.7
    88.2 3244.03   108.8 3242.04   127.7 3238.72   155.9  3238.8   164.6 3236.82
  182.32 3231.52   190.4 3230.09   220.5 3229.84   234.23231.518   237.8 3233.04
   250.2 3241.19     255 3242.44     261    3242   272.1    3243   285.3 3243.07
   302.5  3244.1   311.1 3243.84   341.4 3246.35   376.4 3248.38   422.4  3253.4
   430.3 3254.79   453.8 3256.45   488.3 3263.16   505.6  3265.8   516.1 3269.19
#Mann= 5 ,-1,0
       0      .1       0      30     .06       0  127.71      .1       0
  182.32    .045       0   234.2      .1       0
Bank Sta=182.32,234.2
XS Rating Curve= 0 ,0
Exp/Cntr(USF)=0,0
Exp/Cntr=0.3,0.1

Type RM Length L Ch R = 1 ,3439    ,357.2,377.1,398.3
XS GIS Cut Line= 4
2164502.02982024461136.3606805162164332.08807243461381.276728835
 2164303.3479239461546.220189948 2164288.3530638461597.452628627
#Sta/Elev= 30
       0 3248.75    19.2 3240.68    25.3 3239.03    56.5 3238.67     113  3239.6
   128.4 3238.69   145.6 3239.23   151.9 3238.62   166.5 3239.63   176.3 3238.54
     186 3235.83   200.6 3234.04   262.9  3232.9   288.2 3231.85   297.9 3230.19
   346.7 3231.01   358.9 3227.98   383.3 3227.61  394.813223.927   406.3 3222.84
   440.1 3222.77   444.2 3223.02  446.423223.925   450.1 3226.13   464.5 3238.32
   473.7 3247.45   489.8 3261.96   502.7 3272.72   512.4 3279.85   518.9 3285.93
#Mann= 4 ,-1,0
       0     .06       0     120      .1       0  394.81    .045       0
  446.42      .1       0
Bank Sta=394.81,446.42
XS Rating Curve= 0 ,0
Exp/Cntr(USF)=0,0
Exp/Cntr=0.3,0.1

Type RM Length L Ch R = 1 ,3062    ,202.5,205.4,203.1
XS GIS Cut Line= 4
2164347.08293253461010.1539413322164115.91217264461190.092262545
2163989.70543345461300.0545699542163958.46614158461326.295575131
#Sta/Elev= 30
       0 3237.93    11.4 3235.97    29.9 3235.82    49.8 3233.72    74.7 3234.35
    89.6 3233.79   105.1 3231.09   115.6 3228.43   125.3 3227.22   174.2 3226.92
   223.7 3230.54   239.4 3230.31   252.2 3227.18   267.3  3225.9   297.8  3226.2
   313.8 3227.76   326.1 3227.26   345.7 3228.04   364.6 3222.89   377.5 3222.08
   386.63218.369   391.3 3216.68   399.8 3215.89   422.5 3216.13  434.273218.366
   441.1 3222.39   456.5 3237.05   474.5 3250.59   493.5 3267.16   501.1 3275.83
#Mann= 6 ,-1,0
       0     .06       0      40      .1       0      50     .06       0
     160      .1       0   386.6    .045       0  434.27      .1       0
Bank Sta=386.6,434.27
XS Rating Curve= 0 ,0
Exp/Cntr(USF)=0,0
Exp/Cntr=0.3,0.1

Type RM Length L Ch R = 1 ,2856    ,224.5,228.1,231.4
XS GIS Cut Line= 4
2164137.15489112460908.9386356492163974.71057335461046.391519909
2163849.75340584461153.8546839682163822.26282899461171.348687419
#Sta/Elev= 30
       0 3232.55    12.8 3229.52    37.5  3228.1    56.1 3228.14    60.5 3227.33
    68.5 3224.52    95.6 3222.84   111.6 3223.02   136.6 3222.01   142.8 3222.37
   154.1 3225.03   158.5 3225.28   173.8 3221.41   179.7 3221.07   200.4 3220.99
   250.6 3223.01   274.2 3219.64  286.253216.167     296 3214.82   324.4 3214.93
  332.373216.167   337.5 3218.46     347 3226.22   355.6 3231.34   364.3 3238.02
   374.4  3242.8   389.8 3252.84   398.4 3257.03   406.1  3258.8   410.2 3261.21
#Mann= 5 ,-1,0
       0      .1       0      50     .06       0     200      .1       0
  286.25    .045       0  332.37      .1       0
#XS Ineff= 2 , 0
          249.17 3226.91
Permanent Ineff=
       F       F
Bank Sta=286.25,332.37
XS Rating Curve= 0 ,0
Exp/Cntr(USF)=0,0
Exp/Cntr=0.3,0.1

Type RM Length L Ch R = 1 ,2628    ,219.7,222.5,224.2
XS GIS Cut Line= 4
2163925.97727802460816.4703316922163819.76368564460890.195060522
2163721.04752331460956.4223593022163681.06122971460981.413792804
#Sta/Elev= 30
       0 3227.39     7.1  3225.6    16.2 3223.98    36.3 3223.07    56.4 3220.36
      65 3220.85    73.7  3220.4    89.8 3218.12   113.5 3217.54   120.5 3218.91
   127.5 3219.34   133.6 3219.12   142.7 3218.03   157.7 3218.26   162.9 3217.44
  171.363213.191   177.7 3211.71   194.6 3211.24   215.5 3211.49  220.383213.191
   226.3 3218.29   234.8 3223.74   240.7  3230.3   253.9 3246.23   257.1 3249.58
   263.9 3255.27   272.2  3263.6   277.5 3267.86     290 3275.14   295.3  3278.8
#Mann= 4 ,-1,0
       0     .06       0     120      .1       0  171.36    .045       0
  220.38      .1       0
#XS Ineff= 2 , 0
          155.45 3222.09
Permanent Ineff=
       F       F
Bank Sta=171.36,220.38
XS Rating Curve= 0 ,0
Exp/Cntr(USF)=0,0
Exp/Cntr=0.3,0.1

Type RM Length L Ch R = 1 ,2406    ,187.7,191.8,195.6
XS GIS Cut Line= 4
2163814.76539894460644.0294405282163712.30052158460702.759309258
2163588.59292575460772.7353230632163563.60149225460783.981468139
#Sta/Elev= 30
       0 3228.78    10.4 3227.26    29.1 3225.03    49.1 3223.63    82.7 3220.57
    96.5 3219.66    99.8  3219.2   113.6 3216.36   118.2 3215.73   122.9 3215.75
   127.4  3216.2   136.6 3215.92   150.4 3212.93  159.443209.856   173.4 3208.72
   196.4 3208.79   202.2 3209.15  206.283209.854   214.8  3212.5   219.4 3215.68
   228.5 3226.35   234.4 3232.11   243.3 3238.54   246.9 3241.46   260.9 3251.32
   263.9 3253.59   266.9 3256.25   273.8 3261.73   282.6 3267.76287.6354 3270.95
#Mann= 4 ,-1,0
       0     .06       0  159.44    .045       0  206.28     .06       0
   218.1      .1       0
#XS Ineff= 2 , 0
          130.69 3219.52
Permanent Ineff=
       F       F
Bank Sta=159.44,206.28
XS Rating Curve= 0 ,0
Exp/Cntr(USF)=0,0
Exp/Cntr=0.3,0.1

Type RM Length L Ch R = 1 ,2214    ,189.9,194.2,196.3
XS GIS Cut Line= 4
2163721.04752331460504.0774129182163647.32279448460532.817561445
2163519.86648362460582.8004284492163471.13318829460599.044860225
#Sta/Elev= 30
       0 3222.92     9.5 3218.06    13.9 3216.62    22.4 3214.97      31 3214.16
    39.6 3214.54    52.5 3213.58    78.2 3213.36    86.8 3212.02    95.4 3212.87
   112.6 3212.14   116.9 3211.15   125.5 3207.16  130.983205.374   140.5 3204.07
   151.3 3203.61   165.2 3203.66   168.3 3203.94  172.933205.375     177 3207.42
   181.3 3210.66   202.8 3223.16   211.3 3230.72   224.1 3243.69   230.3 3249.04
   236.6 3253.86     241 3256.32   249.4 3259.89   257.9  3261.5267.4045 3266.23
#Mann= 5 ,-1,0
       0      .1       0   99.13     .06       0  119.13      .1       0
  130.98    .045       0  172.93      .1       0
Bank Sta=130.98,172.93
XS Rating Curve= 0 ,0
Exp/Cntr(USF)=0,0
Exp/Cntr=0.3,0.1

Type RM Length L Ch R = 1 ,2020    ,184.8,181.7,180
XS GIS Cut Line= 4
2163679.81165803 460342.882666832163597.33992747460356.627955256
2163468.63404494460389.1168188092163426.14860799 460404.11167891
#Sta/Elev= 30
       0 3214.79     7.7  3210.5    11.8 3208.76    15.9 3207.33    19.9 3206.84
      24 3206.81    39.9 3209.26    48.3  3209.8    60.5 3210.33    68.6 3209.76
    76.7 3210.04    93.1 3208.78  122.24  3202.7   131.1 3201.57   142.6 3201.25
   163.2 3202.01  167.883202.703   171.4 3204.57   179.7 3215.65   187.9 3222.92
   192.1 3224.98   196.2 3226.43   213.5 3237.14   216.5 3238.64   221.1 3240.26
   233.8 3246.31   242.3    3252   246.5 3253.72     255 3256.35261.4064  3259.4
#Mann= 4 ,-1,0
       0      .1       0      50     .06       0  122.24    .045       0
  167.88      .1       0
#XS Ineff= 2 , 0
           81.85 3212.55
Permanent Ineff=
       F       F
Bank Sta=122.24,167.88
XS Rating Curve= 0 ,0
Exp/Cntr(USF)=0,0
Exp/Cntr=0.3,0.1

Type RM Length L Ch R = 1 ,1838    ,153.3,155.2,156.3
XS GIS Cut Line= 4
2163648.57236615460145.4503421652163549.85620382460177.939205717
2163414.90246291460221.6742143462163358.67173753460239.168217797
#Sta/Elev= 30
       0 3214.04     8.8 3208.37    13.1 3205.93    17.3 3204.05    22.3 3202.66
    29.9 3202.13    42.5 3202.08    76.2 3205.72    93.1 3204.56   101.5 3204.59
   105.7 3204.11   117.4 3201.15   123.8 3199.19   126.7  3198.5   130.9 3198.16
   160.4 3198.12     173 3198.33   177.2  3198.7  179.28 3199.19   198.2 3204.49
   222.2 3205.97     236 3208.29   240.2  3210.2   244.5 3213.37   248.6 3217.01
     257 3222.86   269.6  3230.2   282.7 3240.39   295.5 3247.83304.6777 3253.91
#Mann= 4 ,-1,0
       0      .1       0      20     .06       0   123.8    .045       0
  179.28      .1       0
#XS Ineff= 2 , 0
           77.78 3208.77
Permanent Ineff=
       F       F
Bank Sta=123.8,179.28
XS Rating Curve= 0 ,0
Exp/Cntr(USF)=0,0
Exp/Cntr=0.3,0.1

Type RM Length L Ch R = 1 ,1683    ,158.5,159.3,160
XS GIS Cut Line= 4
 2163596.0903558459994.2521694782163528.61348534460025.491461356
2163391.16060108460064.228183284 2163304.9401555460090.469188461
#Sta/Elev= 30
       0  3221.5    23.2 3207.37    32.3 3203.24    41.3 3200.13    48.4 3199.12
    62.4 3200.79    87.3 3199.65   103.9 3196.06  109.44 3195.37   128.8 3194.25
   145.5 3194.06   153.8 3194.62  156.72 3195.37   162.2  3197.2   182.9 3202.51
     187 3202.17   195.3 3202.58     212 3202.28   224.5 3201.08   228.6 3201.14
   232.8 3201.86     237 3203.81   241.2 3206.41   249.6 3212.85   261.6 3223.45
   266.3 3226.66   278.8 3232.78   287.6 3239.22   297.3 3243.31307.2896 3249.54
#Mann= 4 ,-1,0
       0     .06       0      70      .1       0  109.44    .045       0
  156.72      .1       0
#XS Ineff= 2 , 0
           62.54 3203.79  182.89         3205.45
Permanent Ineff=
       F       F
Bank Sta=109.44,156.72
XS Rating Curve= 0 ,0
Exp/Cntr(USF)=0,0
Exp/Cntr=0.3,0.1

Type RM Length L Ch R = 1 ,1523    ,156.8,156.8,154.9
XS GIS Cut Line= 4
2163548.60663215459856.7992852182163497.37419347459870.544573644
2163353.67345083459908.0317238972163262.45471855459935.522300749
#Sta/Elev= 30
       0 3216.82    13.7 3205.19    21.2 3200.63    29.4 3196.95    33.6 3196.27
    58.4 3195.15    70.8    3195    82.4 3195.35    91.5 3191.52   93.053191.198
    95.6 3190.68     108 3189.79   128.7 3190.02  132.823191.197   144.7 3194.69
   149.4 3197.41   157.6 3198.81   165.9 3198.85   178.3 3198.02   190.9 3198.25
   203.7 3197.59   211.5 3196.66   215.7 3197.05   232.4 3203.31   249.1 3210.61
   258.3 3216.11     270 3221.31   274.1 3224.33   278.3  3226.7296.8253 3235.08
#Mann= 4 ,-1,0
       0     .06       0   93.05    .045       0  132.82     .06       0
  221.55      .1       0
#XS Ineff= 2 , 0
                          159.74         3201.45
Permanent Ineff=
       F       F
Bank Sta=93.05,132.82
XS Rating Curve= 0 ,0
Exp/Cntr(USF)=0,0
Exp/Cntr=0.3,0.1

Type RM Length L Ch R = 1 ,1367    ,198.1,188.8,181.2
XS GIS Cut Line= 4
2163504.87162352459710.5993992312163458.63747154459719.346400957
2163336.17944738 459754.334407862163206.22399317459806.816418214
#Sta/Elev= 30
       0 3212.29    12.9 3203.52    25.1 3196.63    33.3 3194.08    41.4 3192.27
    57.9 3191.53    62.1 3190.91   69.843188.429    76.4 3187.46    97.4 3186.95
   108.8 3187.33   116.2 3188.42   124.9  3193.6   132.8 3195.41     137 3195.62
   145.3 3194.53   157.8 3194.78     182 3193.81   191.7 3194.13   201.2 3193.31
   216.5 3193.83   230.5 3193.29   239.1 3192.23   247.3 3192.51   260.7 3194.24
   273.6 3199.13   282.3 3205.07   287.2 3207.67   303.8 3215.37314.5653 3221.41
#Mann= 4 ,-1,0
       0      .1       0   69.84    .045       0   116.2     .06       0
  184.41      .1       0
#XS Ineff= 2 , 0
                          137.46          3197.3
Permanent Ineff=
       F       F
Bank Sta=69.84,116.2
XS Rating Curve= 0 ,0
Exp/Cntr(USF)=0,0
Exp/Cntr=0.3,0.1
